--- LAURELCK3.prj (project) ---

Proj Title=LAURELCK3
Current Plan=p01
Default Exp/Contr=0,0
English Units
Geom File=g01
Flow File=f01
Plan File=p01
BEGIN DESCRIPTION:
Stream Name: Laurel Creek (I)
Flood Zone: Approximate
Monroe County, West Virginia
HEC-RAS Version: 5.0.7
Vertical Datum: NAVD88
Projection: NAD 1983 StatePlane West Virginia S FIPS 4702 (US Feet)
LiDAR: 2016, 1-meter
Land Use: 2016 NLCD
Hydrologic Method:
SIR2010-5033 regression equations
END DESCRIPTION:
DSS File=dss
DSS Export Rating Curves= 0
DSS Export Rating Curve Sorted= 0
DSS Export Volume Flow Curves= 0
DXF OffsetX= 0
DXF OffsetY= 0
DXF ScaleX= 0
DXF ScaleY= 0

--- LAURELCK3.p01 (plan) ---

Plan Title=Floodplain
Program Version=5.07
Short Identifier=Floodplain
Geom File=g01
Flow File=f01
Subcritical Flow
K Sum by GR= 0
Std Step Tol= 0.01
Critical Tol= 0.01
Num of Std Step Trials= 20
Max Error Tol= 0.3
Flow Tol Ratio= 0.001
Split Flow NTrial= 30
Split Flow Tol= 0.02
Split Flow Ratio= 0.02
Log Output Level= 0
Friction Slope Method= 1
Unsteady Friction Slope Method= 2
Unsteady Bridges Friction Slope Method= 1
Parabolic Critical Depth
Global Vel Dist= 0 , 0 , 0
Global Log Level= 0
CheckData=True
Encroach Param=-1 ,0,0, 0
Computation Interval=0.1SEC
Output Interval=1MIN
Instantaneous Interval=Max Profile
Mapping Interval=1HOUR
Computation Time Step Use Courant=        0
Computation Time Step Use Time Series=    0
Computation Time Step Count To Double=0
Computation Time Step Max Doubling=0
Computation Time Step Max Halving=0
Computation Time Step Residence Courant=0
Run HTab= 0
Run UNet= 0
Run Sediment= 0
Run PostProcess= 0
Run WQNet= 0
Run RASMapper= 0
UNET Theta= 0
UNET Theta Warmup= 0
UNET ZTol= 0
UNET ZSATol= 0
UNET MxIter= 0
UNET Max Iter WO Improvement= 0
UNET MaxInSteps= 0
UNET DtIC= 0
UNET DtMin= 0
UNET MaxCRTS= 0
UNET WFStab= 0
UNET SFStab= 0
UNET WFX= 1
UNET SFX= 1
UNET 1D Methodology=Finite Difference
UNET DSS MLevel= 1
UNET Pardiso=0
UNET DZMax Abort= 0
UNET Use Existing IB Tables= 0
UNET Froude Reduction=False
UNET Froude Limit= 0
UNET Froude Power= 0
UNET D1 Cores= 0
UNET D2 Coriolis=0
UNET D2 Cores= 0
UNET D2 Theta= 1
UNET D2 Theta Warmup= 1
UNET D2 Z Tol= 0.01
UNET D2 Volume Tol= 0.01
UNET D2 Max Iterations= 20
UNET D2 Equation= 0
UNET D2 RampUpFraction=0.1
UNET D2 TimeSlices= 1
UNET D2 BCVolumeCheck=0
UNET D1D2 MaxIter= 0
UNET D1D2 ZTol=0.01
UNET D1D2 QTol=0.1
UNET D1D2 MinQTol=1
DSS File=dss
Write IC File= 0
Write IC File at Fixed DateTime=0
Write IC File at Sim End=0
Echo Input=False
Echo Parameters=False
Echo Output=False
Write Detailed= 0
HDF Write Warmup=0
HDF Write Time Slices=0
HDF Flush=0
HDF Face Node Velocities=0
HDF Compression= 1
HDF Chunk Size= 1
HDF Spatial Parts= 1
HDF Use Max Rows=0
HDF Fixed Rows= 1
Calibration Method= 0
Calibration Iterations= 20
Calibration Max Change=0.05
Calibration Tolerance=0.2
Calibration Maximum=1.5
Calibration Minimum=0.5
Calibration Optimization Method= 1
WQ AD Non Conservative
WQ ULTIMATE=-1
WQ Max Comp Step=1HOUR
WQ Output Interval=15MIN
WQ Output Selected Increments= 0
WQ Output face flow=0
WQ Output face velocity=0
WQ Output face area=0
WQ Output face dispersion=0
WQ Output cell volume=0
WQ Output cell surface area=0
WQ Output cell continuity=0
WQ Output cumulative cell continuity=0
WQ Output face conc=0
WQ Output face dconc_dx=0
WQ Output face courant=0
WQ Output face peclet=0
WQ Output face adv mass=0
WQ Output face disp mass=0
WQ Output cell mass=0
WQ Output cell source sink temp=0
WQ Output nsm pathways=0
WQ Output nsm derived pathways=0
WQ Output MaxMinRange=-1
WQ Daily Max Min Mean=-1
WQ Daily Range=0
WQ Daily Time=0
WQ Create Restart=0
WQ Fixed Restart=0
WQ System Summary=0
WQ Write To DSS=0
WQ Use Fixed Temperature=0
Sorting and Armoring Iterations= 10
XS Update Threshold= 0.02
Bed Roughness Predictor= 0
Hydraulics Update Threshold= 0.02
Energy Slope Method= 1
Volume Change Method= 1
Sediment Retention Method= 0
XS Weighting Method= 0
Number of US Weighted Cross Sections= 1
Number of DS Weighted Cross Sections= 1
Upstream XS Weight=0
Main XS Weight=1
Downstream XS Weight=0
Number of DS XS's Weighted with US Boundary= 1
Upstream Boundary Weight= 1
Weight of XSs Associated with US Boundary= 0
Number of US XS's Weighted with DS Boundary= 1
Downstream Boundary Weight= 0.5
Weight of XSs Associated with DS Boundary= 0.5
Percentile Method= 0
Sediment Output Level= 3
Mass or Volume Output= 0
Output Increment Type= 1
Profile and TS Output Increment= 1
XS Output Flag= 0
XS Output Increment= 10
Write Gradation File= 0
Read Gradation Hotstart= 0
Write HDF5 File= 1
Write Binary Output= 1
Write DSS Sediment File= 0
SV Curve= 0
Specific Gage Flag= 0

--- LAURELCK3.f01 (steady flow) ---

Flow Title=Flow
Program Version=5.07
Number of Profiles= 6
Profile Names=01pct,10pct,04pct,02pct,0_2pct,01plus
River Rch & RM=LAURELCK3,Main            ,44935
     627     332     441     531     874     927
River Rch & RM=LAURELCK3,Main            ,43185
     682     363     481     579     950    1010
River Rch & RM=LAURELCK3,Main            ,42214
     757     405     535     643    1050    1120
River Rch & RM=LAURELCK3,Main            ,41082
     824     441     583     700    1140    1220
River Rch & RM=LAURELCK3,Main            ,38414
     882     474     625     749    1220    1300
River Rch & RM=LAURELCK3,Main            ,37978
     920     495     653     782    1270    1360
River Rch & RM=LAURELCK3,Main            ,37302
    1430     785    1030    1220    1970    2120
River Rch & RM=LAURELCK3,Main            ,36835
    1510     830    1080    1290    2070    2240
River Rch & RM=LAURELCK3,Main            ,34782
    1630     895    1170    1390    2230    2410
River Rch & RM=LAURELCK3,Main            ,29528
    1950    1080    1410    1670    2660    2890
River Rch & RM=LAURELCK3,Main            ,29278
    2040    1130    1470    1750    2790    3020
River Rch & RM=LAURELCK3,Main            ,26368
    2270    1260    1640    1940    3090    3360
River Rch & RM=LAURELCK3,Main            ,22861
    2500    1400    1810    2140    3400    3700
River Rch & RM=LAURELCK3,Main            ,16214
    2670    1500    1930    2290    3620    3950
River Rch & RM=LAURELCK3,Main            ,11315
    2960    1670    2150    2540    4010    4380
Boundary for River Rch & Prof#=LAURELCK3,Main            , 1
Up Type= 0
Dn Type= 3
Dn Slope=0.010546
DSS Import GetInterval= 0
DSS Import GetPeak= 0
DSS Import FillOption= 0

--- LAURELCK3.g01 (geometry) ---

Geom Title=Geometry
Program Version=5.07

River Reach=LAURELCK3       ,Main
Reach XY= 30
     2158128.923      245996.101     2156534.305       241866.76
     2155404.965      240628.045     2154406.701      240364.156
     2154102.882      240647.142     2151174.468      240517.046
     2150587.604      241099.226     2148598.888      244587.941
     2148183.958      244732.906     2147646.631      245629.608
     2146751.666      245737.246     2145875.798      244828.392
     2144578.923      244330.129     2144131.007      243870.927
     2144645.763       242195.58     2145347.152      241848.358
     2145304.618      241580.128     2144644.028      241310.163
     2144379.271      240771.969     2143510.347      240778.045
     2142456.653      239420.564     2142033.784      239267.628
     2141460.868       237231.17     2140466.076      236613.983
     2138148.335      236325.913     2137016.391       235363.24
     2135929.585      235406.642     2133876.633      236554.212
     2131573.248      237150.566     2131110.756      238554.121

Type RM Length L Ch R = 1 ,44935   ,350,350,350
XS GIS Cut Line= 3
     2158514.913      245724.808     2158121.526      245989.398
     2157772.602      246275.753
#Sta/Elev= 30
       0  2538.5    17.5 2537.96    29.2 2543.69    41.1 2545.76    62.4  2546.8
   100.4 2546.46     138 2543.18   191.3  2533.4   199.2 2530.12     219 2530.83
   226.9 2529.34   329.7 2521.78   452.3 2519.65   461.9 2518.16     469 2514.93
   473.7 2513.89   478.4  2515.2   484.6 2519.03   488.9 2519.58   501.6 2518.99
   522.8 2515.72   563.8 2518.88   681.2 2519.74   688.2 2521.77   699.8 2529.66
   704.5 2531.32   725.5 2534.05   744.9 2538.24   798.7 2555.66   925.5 2590.36
#Mann= 6 ,-1 , 0
       0      .1       0      80     .04       0     200    .035       0
     440      .1       0     469    .045       0   478.4      .1       0
Bank Sta=469,478.4
XS Rating Curve= 0 ,0
Exp/Cntr=0.3,0.1

Type RM Length L Ch R = 1 ,44585   ,353.4,350.2,346.9
XS GIS Cut Line= 3
     2158471.169      245570.352     2158027.259      245665.474
     2157572.546      245739.756
#Sta/Elev= 30
       0 2590.45    57.2 2576.07    87.4 2566.94   127.7 2549.79   141.1 2544.88
   167.9    2538     178 2532.27   198.1 2532.46   214.9 2529.38   229.7 2528.31
   301.6 2526.41   349.1 2519.43   409.5 2515.77   436.4 2514.99   446.4 2512.76
   449.8 2511.59   456.5 2511.11   462.1 2512.82   470.7 2514.76   499.7  2514.2
   552.9  2515.9     626 2515.64   639.4 2516.59   695.8 2523.81   712.4 2527.69
   732.4 2534.93   788.9 2561.52   812.2 2570.18     862 2581.72   914.7 2591.98
#Mann= 7 ,-1 , 0
       0      .1       0      30     .04       0     330    .035       0
   446.4    .045       0   462.1    .035       0  633.99     .12       0
  733.99      .1       0
#XS Ineff= 2 , 0
                          563.16          2516.5
Permanent Ineff=
       F       F
Bank Sta=446.4,462.1
XS Rating Curve= 0 ,0
Exp/Cntr=0.3,0.1

Type RM Length L Ch R = 1 ,44235   ,203.2,200.5,197.8
XS GIS Cut Line= 3
     2158338.079      245118.005     2157936.083      245330.825
     2157519.856      245516.646
#Sta/Elev= 30
       0 2587.52    31.5  2580.3    56.9 2571.81     128 2543.14   135.4 2539.31
   142.9 2533.25   165.1 2532.86   168.8 2531.99     180  2525.5   194.8 2522.37
   261.7 2516.84   287.2 2513.33   309.9 2511.56   395.3  2510.4   435.5 2512.43
   439.8 2512.02     4452509.986   448.5 2509.04   458.22509.859   476.3 2511.86
   627.2 2512.08   638.8 2512.82   656.2 2515.88   678.5 2522.33   720.6 2531.98
   760.1 2546.28   785.2 2558.78   806.8 2565.47   839.1 2571.66   910.7 2577.95
#Mann= 8 ,-1 , 0
       0      .1       0     100     .04       0     210    .035       0
     445    .045       0   458.2    .035       0  654.86      .1       0
  814.86     .12       0  864.86      .1       0
#XS Ineff= 2 , 0
          434.96 2512.72  572.37         2513.48
Permanent Ineff=
       F       F
Bank Sta=445,458.2
XS Rating Curve= 0 ,0
Exp/Cntr=0.3,0.1

Type RM Length L Ch R = 1 ,44034   ,81,81,80.9
XS GIS Cut Line= 2
2158183.91181766 244874.317562962157504.94354352245432.229478144
#Sta/Elev= 30
       0 2528.65    14.8  2524.9    36.1 2520.71   150.9 2517.87   193.2 2515.97
   204.5 2514.73   231.4 2509.72   239.5 2509.18   346.1 2508.58   386.3 2509.55
   405.5 2508.35   425.9  2509.9   440.5 2507.47   449.2 2505.94   452.2  2506.1
   455.32507.383   465.6  2510.1   507.4 2509.34   562.6 2511.16   571.1 2510.89
   588.1 2512.05   610.1 2516.75   639.1 2526.15   664.5 2537.13     680 2542.64
   693.7 2545.96   709.2 2548.71   770.7 2555.69   802.2 2558.62   878.8 2562.06
#Mann= 9 ,-1 , 0
       0     .04       0      40    .035       0     430     .06       0
   440.5    .045       0   455.3     .06       0     490    .035       0
     680     .12       0     800      .1       0     810     .12       0
Bank Sta=440.5,455.3
XS Rating Curve= 0 ,0
Exp/Cntr(USF)=0,0
Exp/Cntr=0.5,0.3

Type RM Length L Ch R = 1 ,43953   ,42.9,42.9,42.8
XS GIS Cut Line= 2
     2158146.054      244799.485      2157455.95      245369.146
#Sta/Elev= 30
       0 2521.97    97.9 2520.25     204 2516.27   221.4 2515.26   256.3 2510.76
   284.3  2510.2   314.8 2508.03   402.2 2507.53   446.5 2509.51   456.72507.366
   463.8 2506.13   470.62507.398   479.5 2509.71   510.4 2509.46   540.1 2510.45
     562 2514.01   575.6 2513.48   603.6 2521.71   615.2 2526.01   625.2 2527.27
   637.9 2532.37   646.4 2534.48   687.5 2537.08     706 2540.02   722.4 2541.58
   752.8 2542.33   778.3 2540.71     797 2540.58   850.6 2543.73   894.9 2545.25
#Mann= 8 ,-1 , 0
       0    .035       0     450     .06       0   456.7    .045       0
   470.6     .06       0     510    .035       0     630      .1       0
     760     .12       0     890      .1       0
#XS Ineff= 2 , 0
             435  2510.5     495          2510.5
Permanent Ineff=
       F       F
Bank Sta=456.7,470.6
XS Rating Curve= 0 ,0
Exp/Cntr=0.5,0.3

Type RM Length L Ch R = 1 ,43910   ,99,98.8,98.8
XS GIS Cut Line= 2
     2158115.672      244769.103     2157425.568      245338.764
#Sta/Elev= 30
       0 2520.08   207.4 2516.11   254.1 2511.79   313.5 2510.71   362.3 2507.08
   429.3 2507.55   442.8 2509.06   449.6 2507.14   458.2 2505.19   464.8  2507.3
   477.7 2509.57   505.7 2510.91   554.6 2510.98   568.8 2515.78   577.3 2521.69
     590 2526.38     620 2531.86   649.6 2533.48   662.4 2533.33   673.5 2528.74
   682.8 2527.52   717.9 2532.76   738.5 2533.43   785.7 2531.17   808.7 2523.53
   819.8  2524.5   836.6 2529.16   848.3 2529.84   879.3 2522.26   894.9 2521.51
#Mann= 8 ,-1 , 0
       0    .035       0   449.6    .045       0   464.8    .035       0
     470     .06       0     500    .035       0     590      .1       0
     810     .12       0     850      .1       0
#XS Ineff= 2 , 0
           446.7  2510.5   473.3          2510.5
Permanent Ineff=
       F       F
Bank Sta=449.6,464.8
XS Rating Curve= 0 ,0
Exp/Cntr=0.5,0.3

Type RM Length L Ch R = 1 ,43812   ,269.4,276.4,280.5
XS GIS Cut Line= 3
2158111.53697219244742.6702389762157894.43848481244818.206036255
2157373.36054465245265.557679583
#Sta/Elev= 30
       0 2519.94    84.9 2517.95   156.7 2514.96   203.1 2513.84   231.6 2512.52
   278.6  2511.2   303.4 2510.95   327.3    2510   337.3 2509.02     365  2507.4
   382.5 2507.66   402.8  2506.9   434.2 2506.85   455.8 2507.36   468.6 2505.78
   473.3 2504.05   477.5 2504.42  480.98 2505.85   486.1 2507.59   490.4 2508.22
   512.1 2509.17   543.8 2509.23   585.6 2510.25   615.8 2509.13     672 2514.36
   693.7 2514.79   735.2  2514.4   833.8 2517.68   886.3 2520.16   916.6 2520.97
#Mann= 8 ,-1 , 0
       0    .035       0   468.6    .045       0  480.98    .035       0
  489.86     .06       0  539.86    .035       0  639.86      .1       0
  669.86    .035       0  789.86      .1       0
Bank Sta=468.6,480.98
XS Rating Curve= 0 ,0
Exp/Cntr(USF)=0,0
Exp/Cntr=0.3,0.1

Type RM Length L Ch R = 1 ,43535   ,348.5,350.3,349.7
XS GIS Cut Line= 3
     2157984.342      244576.377      2157565.31      244756.775
     2157120.685      244866.793
#Sta/Elev= 30
       0 2517.74     209 2511.09   316.4 2506.66   391.7 2505.62   433.7 2505.51
   438.2 2505.26   445.3 2503.85   452.4 2503.07   462.8  2502.3   466.2 2502.52
  468.09 2503.12   479.7  2505.9     486 2510.57   494.2 2518.22   506.7 2527.58
   510.4 2530.23   516.9 2533.54   537.1  2538.9   567.6 2545.38   594.6 2551.84
   635.3  2558.4   652.1 2560.35   672.3 2562.09   709.5 2563.39   724.5  2564.6
   765.1 2570.66   807.5 2578.12   827.8 2580.47     865 2582.61   914.2 2588.15
#Mann= 7 ,-1 , 0
       0    .035       0     360      .1       0   452.4    .045       0
  468.09     .12       0  566.21      .1       0  586.21     .12       0
  666.21      .1       0
#XS Ineff= 2 , 0
           362.9 2506.91
Permanent Ineff=
       F       F
Bank Sta=452.4,468.09
XS Rating Curve= 0 ,0
Exp/Cntr=0.3,0.1

Type RM Length L Ch R = 1 ,43185   ,351.7,350.2,347.6
XS GIS Cut Line= 3
     2157934.459      244295.883     2157496.488      244417.875
     2157052.929      244530.857
#Sta/Elev= 30
       0 2514.56    32.2 2512.14    86.7    2510   178.7 2508.08   253.6 2507.59
   284.2  2505.8   314.9 2502.68     383 2502.72   396.9 2501.81   434.1 2503.04
   444.3 2500.41   451.1 2499.23   458.62500.297   464.7  2501.5   488.4 2503.31
   501.9 2507.15   512.6 2507.78   539.2 2518.72   559.5 2528.27   566.1 2530.68
   576.4 2532.92   593.3 2534.42   627.2 2535.86   674.1 2536.25   749.1 2543.44
   772.8  2544.8   813.4 2550.09   837.1 2555.46   858.1 2559.13   912.4 2564.27
#Mann= 6 ,-1 , 0
       0    .035       0     290      .1       0     370    .035       0
     390      .1       0   444.3    .045       0   458.6      .1       0
Bank Sta=444.3,458.6
XS Rating Curve= 0 ,0
Exp/Cntr=0.3,0.1

Type RM Length L Ch R = 1 ,42835   ,59.7,63.4,68.9
XS GIS Cut Line= 2
2157877.82618793243892.7361407612157052.80893203244259.050285817
#Sta/Elev= 30
       0 2531.87    11.5 2529.18    22.3 2521.58    40.2 2520.54    54.6 2513.46
    76.1 2509.64   181.3 2505.57   220.3 2501.45   247.6 2500.17   294.9 2499.29
   435.1 2499.54   445.8 2499.16     453 2497.75   460.2  2496.4   468.22497.646
   474.6 2498.55   492.5 2497.24   510.4 2498.66   535.6 2498.65   564.3 2500.75
   596.6 2513.91   625.5 2529.93   646.9 2540.64   660.3 2541.38   670.2 2546.18
   700.7 2553.49   786.9 2567.83   809.5 2570.43   857.3 2581.83   902.7  2596.3
#Mann= 5 ,-1 , 0
       0     .04       0     350    .035       0     453    .045       0
   468.2    .035       0     570      .1       0
#XS Ineff= 2 , 0
          323.14  2502.7
Permanent Ineff=
       F       F
Bank Sta=453,468.2
XS Rating Curve= 0 ,0
Exp/Cntr(USF)=0,0
Exp/Cntr=0.5,0.3

Type RM Length L Ch R = 1 ,42771   ,36.1,36.5,35.8
XS GIS Cut Line= 4
2157883.22364856243874.3880163272157457.84539976244021.432349245
2157398.76508743244024.0581409042157028.52846348244247.250431941
#Sta/Elev= 30
       0 2536.89    13.3 2531.84    27.2 2528.23    37.6 2520.09    58.5 2519.33
    65.4 2514.99    72.4 2512.43   100.1 2507.69   214.7 2503.85   256.3 2499.41
   422.7 2498.85   463.9 2500.07   473.3 2496.43   483.5 2495.54   487.9 2496.33
   496.7 2499.54   541.7 2498.39   582.7 2500.84   613.4  2510.7   647.8 2524.25
   655.5 2529.24   670.8 2530.28   686.1 2538.41   709.7 2545.61   746.8 2555.25
   762.7 2557.33   808.7 2566.87   826.1 2568.44   889.2  2585.2   941.5 2602.69
#Mann= 5 ,-1 , 0
       0     .04       0     390    .035       0   473.3    .045       0
   487.9    .035       0  549.21      .1       0
#XS Ineff= 4 ,-1
       0  207.45  2500.5  207.45  336.44 2503.66  336.44     455  2500.5
     505   941.5  2500.5
Permanent Ineff=
       F       F       F       F
Bank Sta=473.3,487.9
XS Rating Curve= 0 ,0
Exp/Cntr(USF)=0,0
Exp/Cntr=0.5,0.3

Type RM Length L Ch R = 1 ,42735   ,117.5,111.8,108
XS GIS Cut Line= 4
2157876.65916942243838.9398289272157451.28092062243985.984161845
2157392.20060828243988.6099535042157021.96398433244211.802244541
#Sta/Elev= 30
       0 2542.44    18.2 2533.84    41.1 2526.48    51.5 2519.02    72.4 2518.06
    84.2 2511.92   110.5 2507.06   228.3  2502.7   277.2 2499.38     440 2499.07
   463.8 2499.74   470.4 2496.15   480.2 2495.01   485.1 2496.09   493.4 2499.83
     575 2498.87   586.5 2501.13   599.4 2499.69   624.8 2510.03   651.1 2518.68
   659.3 2523.19   674.6 2524.02   693.8 2532.92   706.1 2536.88   753.9 2550.13
   801.7    2561   812.5 2564.94   835.2    2568   877.7  2579.7   941.5 2599.93
#Mann= 5 ,-1 , 0
       0     .04       0     440    .035       0   470.4    .045       0
   485.1    .035       0  549.21      .1       0
#XS Ineff= 4 ,-1
       0  237.43  2500.5  237.43  351.63 2501.95  351.63   461.7  2500.5
   488.3   941.5  2500.5
Permanent Ineff=
       F       F       F       F
Bank Sta=470.4,485.1
XS Rating Curve= 0 ,0
Exp/Cntr(USF)=0,0
Exp/Cntr=0.5,0.3

Type RM Length L Ch R = 1 ,42623   ,190.7,182.2,176.8
XS GIS Cut Line= 2
2157819.79813267243693.3140020942156968.82813267244067.391002094
#Sta/Elev= 30
       0    2541    48.4  2527.1    59.2  2522.1    66.3 2521.75      75 2523.07
    88.9 2514.97   105.8 2514.97   127.3 2511.98   253.2 2506.98   263.5 2504.94
   317.2 2498.56   417.4 2497.31   441.9 2498.48     4482495.828   457.4 2493.97
   464.1 2495.69   471.3 2497.78   477.3 2498.17     520 2496.97   572.3 2496.83
     629 2498.43   639.8 2499.98   657.7 2504.39     669 2505.24   678.9 2509.19
   722.2 2521.84   768.8 2541.06   798.4 2554.55   858.2 2576.62   929.6 2608.41
#Mann= 7 ,-1 , 0
       0     .04       0      30      .1       0      70     .04       0
     448    .045       0   464.1     .04       0     520    .035       0
     610      .1       0
#XS Ineff= 2 , 0
          373.67 2500.84  597.07         2501.41
Permanent Ineff=
       F       F
Bank Sta=448,464.1
XS Rating Curve= 0 ,0
Exp/Cntr=0.3,0.1

Type RM Length L Ch R = 1 ,42441   ,216.6,226.2,231.5
XS GIS Cut Line= 4
2157744.86962672243521.3564492392157335.07738971243683.438453426
2157220.39672637243859.2821372142156948.22128538243975.491876065
#Sta/Elev= 30
       0 2510.98    32.3 2509.69   134.6 2508.78     200 2504.87   255.3 2502.32
   273.8 2502.32   432.8 2497.55   457.2 2497.45   484.6 2496.37   490.4 2493.97
   495.2 2493.09   504.6 2494.12   515.9 2495.34   528.4 2495.24   535.5 2496.26
   617.8 2497.11   664.2 2501.57   689.2 2502.94   705.9 2504.62   732.8 2507.83
   751.5 2512.11   767.7 2517.18   806.2  2536.2   814.2 2541.43   839.6 2554.29
   864.6 2568.37   871.7 2571.57   881.8 2577.19   928.2  2599.1   946.6 2608.94
#Mann= 7 ,-1 , 0
       0      .1       0     100     .06       0     200     .04       0
   490.4    .045       0   504.6     .04       0  710.62    .035       0
  760.62      .1       0
Bank Sta=490.4,504.6
XS Rating Curve= 0 ,0
Exp/Cntr(USF)=0,0
Exp/Cntr=0.3,0.1

Type RM Length L Ch R = 1 ,42214   ,171,173.5,171.3
XS GIS Cut Line= 2
     2157652.482      243354.138     2156819.012      243717.277
#Sta/Elev= 30
       0 2525.22    30.2 2521.47    41.2 2515.79    62.7 2516.84   109.2 2514.41
   127.4 2509.45   152.1 2510.11   184.4 2506.61   294.4 2502.89   366.2 2497.07
   491.3  2494.8   511.2 2492.86   520.8 2491.46   528.7  2492.6   556.5 2492.26
   570.9 2494.11   642.4 2492.67   678.3 2511.92   699.7 2519.94   721.2 2529.85
   731.9 2536.92   746.2 2539.45     753 2544.77   760.5 2548.77   803.5 2567.23
   815.3 2574.52   835.7 2578.98     850 2588.51   882.6 2602.44   909.1 2611.91
#Mann= 10 ,-1 , 0
       0     .06       0     100     .04       0     140    .035       0
     210     .04       0     430     .06       0   511.2    .045       0
   528.7     .06       0     530      .1       0     850     .08       0
     880      .1       0
Bank Sta=511.2,528.7
XS Rating Curve= 0 ,0
Exp/Cntr=0.3,0.1

Type RM Length L Ch R = 1 ,42041   ,151.2,153.9,153
XS GIS Cut Line= 2
2157617.33117836243137.1910903572156771.34061202243593.979385127
#Sta/Elev= 30
       0 2568.31    40.3 2558.95   112.6 2536.64   163.3 2518.76   173.1  2516.7
   193.1 2506.05   214.3 2505.74     224 2502.67   245.3 2499.28   301.8 2494.07
   327.4 2492.87   457.9 2492.46   526.6 2493.46   547.3 2492.74   577.2 2493.75
   589.6 2491.86   605.7 2490.87  609.39 2491.94   618.2 2493.65     648 2492.55
   670.4 2493.88   676.8 2495.32   695.4 2502.46     745 2510.36   768.8 2518.88
   826.6 2544.82     868 2560.73     909 2572.41   938.2 2578.52   961.4 2581.85
#Mann= 8 ,-1 , 0
       0      .1       0     160     .04       0     180    .035       0
     370     .04       0     510      .1       0   589.6    .045       0
  609.39      .1       0     850     .08       0
#XS Ineff= 2 , 0
          461.81 2498.03
Permanent Ineff=
       F       F
Bank Sta=589.6,609.39
XS Rating Curve= 0 ,0
Exp/Cntr(USF)=0,0
Exp/Cntr=0.3,0.1

Type RM Length L Ch R = 1 ,41887   ,45.1,45.4,44.7
XS GIS Cut Line= 2
2157524.49896789243014.6268956462156702.01596789243472.525895646
#Sta/Elev= 30
       0 2549.53    28.2 2540.19      62 2530.85    88.1 2524.38   138.9 2513.64
   152.1 2506.14   155.6 2505.06   178.4 2504.83   198.5 2500.48   227.2 2496.51
     250  2495.3     291 2494.93   324.8 2492.41   399.9 2491.09   508.8 2492.27
  526.57 2489.83     532 2489.22   540.82489.767   557.6 2491.89     621 2491.44
   655.1 2493.95   670.3  2496.3   707.8 2506.03   752.9 2513.92     798 2525.03
   816.7 2528.36     843 2530.69     858 2531.32   873.1 2529.89   941.4  2533.7
#Mann= 7 ,-1 , 0
       0      .1       0     190     .04       0  526.57    .045       0
   540.8     .04       0     610      .1       0     750     .08       0
     860      .1       0
Bank Sta=526.57,540.8
XS Rating Curve= 0 ,0
Exp/Cntr=0.5,0.3

Type RM Length L Ch R = 1 ,41842   ,49.2,46.7,46.9
XS GIS Cut Line= 2
     2157511.867      242973.573     2156689.384      243431.472
#Sta/Elev= 30
       0 2561.47     6.2    2560    13.7    2556    37.6 2546.94    73.8  2535.7
    85.1 2533.47   103.8 2526.73   145.3 2511.55   157.4 2504.63   175.2 2504.47
   197.7 2500.23     239 2496.17     290 2495.14   321.6 2493.13   391.3 2491.42
   501.9 2491.95   521.52488.716   528.8 2487.64   534.62488.704   543.2 2490.88
   632.5 2492.65   644.6 2493.93   689.6 2503.75   704.6 2505.86   826.8 2517.34
   839.3 2515.95   854.8 2506.26     881 2502.98   907.5 2504.64   941.4 2511.97
#Mann= 11 ,-1 , 0
       0      .1       0     170     .04       0     280    .035       0
     290     .04       0     400    .035       0     500     .04       0
   521.5    .045       0   534.6     .04       0     700      .1       0
     740     .08       0     850      .1       0
#XS Ineff= 2 , 0
           497.5    2493   562.5            2493
Permanent Ineff=
       F       F
Bank Sta=521.5,534.6
XS Rating Curve= 0 ,0
Exp/Cntr(USF)=0,0
Exp/Cntr=0.5,0.3

Type RM Length L Ch R = 1 ,41795   ,167.5,168.8,169.8
XS GIS Cut Line= 2
2157490.47123732  242940.69909332156667.98823732  243398.5990933
#Sta/Elev= 30
       0 2561.45       9 2559.23    19.3 2553.85    56.8 2539.78    86.2 2531.13
   139.3 2511.68   151.3 2504.56   173.2  2503.3   188.2 2498.84   259.6 2495.23
   342.2 2492.33   413.5 2491.39   466.1 2491.98     477 2491.12   489.7 2488.32
   498.7 2487.38   505.9 2488.23   513.1  2489.4   556.6 2490.76   567.5 2492.52
   635.1 2493.76   661.4 2503.62   672.6 2504.86   732.7 2505.85   766.5 2501.54
   834.1  2502.8   864.2 2500.83   871.7 2504.38   879.2 2505.92   941.4 2506.54
#Mann= 10 ,-1 , 0
       0      .1       0     150     .04       0     260    .035       0
     360     .04       0     370    .035       0   489.7    .045       0
   505.9    .035       0     560     .04       0     770     .08       0
     820      .1       0
#XS Ineff= 2 , 0
           484.2    2493   515.8            2493
Permanent Ineff=
       F       F
Bank Sta=489.7,505.9
XS Rating Curve= 0 ,0
Exp/Cntr(USF)=0,0
Exp/Cntr=0.5,0.3

Type RM Length L Ch R = 1 ,41626   ,243.3,243.2,242.9
XS GIS Cut Line= 3
2157444.68035372  242836.48535822156832.80302698243175.222117276
2156557.45851827243187.013631127
#Sta/Elev= 30
       0 2559.29    25.4 2551.25    44.8 2546.56    64.4 2538.25   129.2 2516.19
   143.2 2512.27   150.7 2508.82   158.2 2503.37   177.5 2503.23   188.2 2499.38
   203.2 2497.28   248.2 2494.88   281.3 2491.48   323.2  2489.3   370.6 2489.95
  380.73 2487.47   386.9 2486.21   394.7 2487.36   401.9 2489.11   414.1 2489.75
     472 2489.46   499.4  2491.2   686.8 2496.29   739.7 2502.86     764 2508.84
   800.8 2527.79   846.1 2553.07   901.9 2576.99   941.4 2595.37     975    2609
#Mann= 8 ,-1 , 0
       0      .1       0     100     .04       0  380.73    .045       0
   394.7     .04       0     550    .035       0     660      .1       0
  759.38     .12       0  959.38      .1       0
Bank Sta=380.73,394.7
XS Rating Curve= 0 ,0
Exp/Cntr=0.3,0.1

Type RM Length L Ch R = 1 ,41383   ,295.9,300.9,301.5
XS GIS Cut Line= 2
2157292.53056028242630.3760602932156518.62758918 243137.21427814
#Sta/Elev= 30
       0  2529.6    28.4 2527.59    52.1 2527.59    81.6 2520.96   101.2 2515.42
   120.8 2505.75   144.3 2505.48     160 2502.02   214.9 2495.75   258.6  2488.3
   277.7 2487.17   405.2 2488.52     4342485.773   443.1 2484.58   450.2 2485.81
   450.2 2485.82   450.2 2485.83   457.3 2487.37   540.3 2487.26     560 2488.25
   604.3 2494.91   630.6 2502.02   668.3 2522.71   694.3 2538.97   710.9 2545.52
   725.1 2555.68   786.7 2589.07     862  2621.9   893.4 2632.04   925.1 2639.33
#Mann= 7 ,-1 , 0
       0      .1       0      30     .04       0     390    .035       0
     434    .045       0   450.2    .035       0     530     .12       0
     740      .1       0
#XS Ineff= 2 , 0
                          522.03         2507.89
Permanent Ineff=
       F       F
Bank Sta=434,450.2
XS Rating Curve= 0 ,0
Exp/Cntr(USF)=0,0
Exp/Cntr=0.3,0.1

Type RM Length L Ch R = 1 ,41082   ,330.3,331,328.6
XS GIS Cut Line= 3
     2157186.665      242451.001     2156748.578      242638.508
     2156337.818      242825.212
#Sta/Elev= 30
       0 2508.71      36 2509.58      56 2508.54    76.8  2505.2    98.3  2500.1
   118.4  2500.4   151.8 2497.62   182.3  2492.7   340.7 2485.85   394.5 2484.74
   455.1 2486.09   465.9 2483.95   480.1 2482.65  485.36 2483.95     491 2486.69
   547.7 2486.73   573.8 2488.43   602.7 2493.37   609.9 2495.45   660.3 2518.03
   711.2 2537.92   736.1 2545.66   750.4 2548.16   768.5 2549.62   782.9 2549.17
   847.7 2544.61   869.4 2547.13   901.8 2537.74     909 2540.01   927.7 2550.74
#Mann= 7 ,-1 , 0
       0      .1       0      20     .06       0     130     .04       0
     190    .035       0   465.9    .045       0  485.36    .035       0
  676.53     .12       0
Bank Sta=465.9,485.36
XS Rating Curve= 0 ,0
Exp/Cntr=0.3,0.1

Type RM Length L Ch R = 1 ,40751   ,26.7,26.7,26.6
XS GIS Cut Line= 2
 2157012.0237711242132.670638591 2156269.8357711242542.827638591
#Sta/Elev= 30
       0  2514.1    19.8 2514.22    64.9 2511.57    75.3 2509.02    87.3 2503.46
   121.2 2500.65   166.1 2492.32   186.4 2486.72   215.3 2484.14     241 2482.74
   271.6 2482.05   357.2 2482.23   394.7 2483.13   415.7 2481.77   424.7 2480.15
   428.5  2480.5   432.3  2481.8     436 2482.59   492.2 2483.75   529.7 2487.25
   600.9 2491.49   615.9 2493.69   631.9  2498.1   659.6 2509.16   702.1 2527.53
   735.8 2538.79   756.1 2544.51   779.3 2549.21   810.8 2557.43     848 2563.25
#Mann= 6 ,-1 , 0
       0     .06       0      50     .04       0     160    .035       0
   415.7    .045       0   432.3    .035       0     610     .12       0
#XS Ineff= 2 , 0
          254.72 2483.97
Permanent Ineff=
       F       F
Bank Sta=415.7,432.3
XS Rating Curve= 0 ,0
Exp/Cntr=0.5,0.3

Type RM Length L Ch R = 1 ,40724   ,52.9,52.8,52.7
XS GIS Cut Line= 2
     2157000.655      242108.512     2156258.467      242518.669
#Sta/Elev= 30
       0 2514.99     6.9 2513.68    29.2 2513.65    63.1 2511.99    78.1 2508.49
    89.5 2502.36      92 2501.73   111.8 2500.53   141.8 2495.49   160.6 2493.28
   175.6 2490.72   198.4 2485.32   210.3 2483.58   318.9 2481.97   404.2 2483.56
   419.12481.201   426.7 2480.04   433.52481.208   444.4 2483.37   456.5 2482.54
   503.7 2483.92   591.8 2489.37   606.6 2491.38   623.1 2495.87   642.4 2503.71
   693.1 2527.47   730.3 2543.52   750.6 2551.22   820.3  2571.9     848 2578.17
#Mann= 7 ,-1 , 0
       0      .1       0      50     .04       0     150    .035       0
   419.1    .045       0   433.5    .035       0     600     .12       0
     820      .1       0
#XS Ineff= 4 ,-1
       0  158.24    2482  158.24  262.54  2489.6  262.54   397.5    2482
   452.5     848    2482
Permanent Ineff=
       F       F       F       F
Bank Sta=419.1,433.5
XS Rating Curve= 0 ,0
Exp/Cntr(USF)=0,0
Exp/Cntr=0.5,0.3

Type RM Length L Ch R = 1 ,40671   ,75.4,75.5,75.6
XS GIS Cut Line= 2
     2156986.549      242056.429     2156244.361      242466.585
#Sta/Elev= 30
       0 2531.74    35.7 2522.65    57.1 2513.88    88.5 2510.74   102.6 2504.15
   107.8 2500.35   110.7 2499.16   129.6 2498.19   160.9  2492.1   217.9 2484.21
   234.4 2483.15   325.1 2481.69     412 2482.61   421.7 2481.91   425.62480.578
   436.8 2479.31   441.8  2480.6   448.5 2482.58   485.6 2482.29   500.6 2483.22
   534.3 2482.62   571.8 2483.93   594.3 2487.04   624.3 2494.44   653.5 2507.25
   673.7 2517.66   704.2 2531.67   757.5 2558.43     820  2587.1     848 2598.68
#Mann= 7 ,-1 , 0
       0      .1       0     130     .04       0     160    .035       0
   425.6    .045       0   441.8    .035       0     580     .12       0
     810      .1       0
#XS Ineff= 4 ,-1
       0  179.34    2482  179.34  306.81 2485.42  306.81   424.2    2482
   445.8     848    2482
Permanent Ineff=
       F       F       F       F
Bank Sta=425.6,441.8
XS Rating Curve= 0 ,0
Exp/Cntr(USF)=0,0
Exp/Cntr=0.5,0.3

Type RM Length L Ch R = 1 ,40596   ,358.6,354.1,347.2
XS GIS Cut Line= 2
2156955.28487947241991.0585661642156213.09687947242401.214566164
#Sta/Elev= 30
       0 2532.93    58.1 2518.81    67.7 2515.01    78.7  2512.6   108.8 2510.37
   115.7 2507.26   127.5 2498.38   131.2 2496.67   149.6 2496.16   161.2 2491.72
   172.5 2490.58   207.8 2483.33   224.7 2481.84   281.2 2480.53   401.1 2482.07
   409.22480.525   416.1 2478.71   424.72480.245   431.1 2482.01   454.8 2482.63
   524.8 2481.37   577.3 2482.55   592.3 2483.23     611 2486.28   632.7 2495.21
   712.2 2537.66   734.1 2547.84   804.1 2582.97   840.3 2602.69     848 2606.14
#Mann= 9 ,-1 , 0
       0      .1       0     100     .04       0     290    .035       0
   409.2    .045       0   424.7    .035       0     550     .12       0
     660      .1       0     700     .12       0     770      .1       0
#XS Ineff= 2 , 0
          310.03 2484.88  497.29         2484.79
Permanent Ineff=
       F       F
Bank Sta=409.2,424.7
XS Rating Curve= 0 ,0
Exp/Cntr=0.3,0.1

Type RM Length L Ch R = 1 ,40242   ,208.2,210,210
XS GIS Cut Line= 3
     2156974.331      241844.705     2156587.128      241779.078
     2156167.112      242260.346
#Sta/Elev= 30
       0 2544.66    65.9 2534.25   149.1 2519.25     229 2510.07   301.2 2499.01
   315.5 2492.13   338.8  2491.6   352.1 2487.64   372.1 2487.56   388.7 2484.28
   401.7 2485.27   421.6 2484.59   434.8 2480.84   475.2 2478.76   484.5 2477.11
   495.8 2475.52   505.4  2477.2   513.2 2478.53   539.3 2480.03   576.3 2478.59
     624 2479.65   722.2 2479.56   742.6 2482.16     803 2485.82   820.8 2488.26
   840.8 2493.47     910 2517.77   985.5 2539.87  1000.7 2546.76  1031.5 2563.61
#Mann= 8 ,-1 , 0
       0      .1       0     310     .04       0  412.73    .035       0
   484.5    .045       0   505.4    .035       0  862.73     .12       0
  992.73      .1       0 1012.73     .12       0
#XS Ineff= 2 , 0
          464.99 2480.73  700.03         2481.24
Permanent Ineff=
       F       F
Bank Sta=484.5,505.4
XS Rating Curve= 0 ,0
Exp/Cntr=0.3,0.1

Type RM Length L Ch R = 1 ,40032   ,137.8,138.2,138.6
XS GIS Cut Line= 3
     2156701.894      241423.089     2156358.856       241724.69
     2156043.033      242051.794
#Sta/Elev= 30
       0 2542.33    69.6 2526.54    78.9 2525.72   120.1    2516     130 2512.42
   147.5 2510.39   164.9 2504.24   195.6 2502.44   217.4  2496.3   239.3 2495.94
   257.9 2491.39   297.4 2487.84   341.6 2485.19   374.7 2485.05     409 2478.33
   427.6 2478.25   448.5 2475.88   457.9  2474.6   463.32475.977   467.2 2477.59
   476.1 2478.46   590.1 2476.68   685.2 2477.93   701.5 2479.11   717.6  2482.1
   729.3 2486.44   760.1 2502.98   818.1 2536.61   854.6 2555.97   911.5  2588.4
#Mann= 8 ,-1 , 0
       0      .1       0      40     .12       0     170    .035       0
     180     .04       0     300    .035       0   448.5    .045       0
   463.3    .035       0  616.77      .1       0
#XS Ineff= 2 , 0
          423.68 2479.45  639.47         2482.25
Permanent Ineff=
       F       F
Bank Sta=448.5,463.3
XS Rating Curve= 0 ,0
Exp/Cntr=0.3,0.1

Type RM Length L Ch R = 1 ,39894   ,176,176,175.2
XS GIS Cut Line= 2
 2156629.7519201241299.3807490692155895.51878644241960.980067359
#Sta/Elev= 30
       0 2537.12    36.4 2532.16     136 2521.68   180.1 2515.14   208.3 2512.16
   229.7 2506.56   237.5 2501.62   240.8 2500.46   261.7 2499.81   284.9 2492.43
     317 2485.49   366.3 2481.54   454.5 2477.48   459.2 2476.87   464.82474.653
   471.6 2473.34   479.7  2474.6   504.2 2477.32   551.1 2476.19   570.7 2476.77
   595.2 2478.96   607.1 2478.03   621.8 2474.22   710.1 2474.75   734.6 2486.53
   823.9 2536.01   886.7 2564.83   917.6  2576.3   970.6 2589.72   988.3 2592.45
#Mann= 7 ,-1 , 0
       0      .1       0     210     .04       0     340    .035       0
   464.8    .045       0   479.7    .035       0     660      .1       0
     740     .05       0
#XS Ineff= 2 , 0
                          598.68            2480
Permanent Ineff=
       F       F
Bank Sta=464.8,479.7
XS Rating Curve= 0 ,0
Exp/Cntr(USF)=0,0
Exp/Cntr=0.3,0.1

Type RM Length L Ch R = 1 ,39718   ,207.1,203.5,198.5
XS GIS Cut Line= 2
 2156456.0623616241209.3779778452155778.67308345241856.766332258
#Sta/Elev= 30
       0 2496.53    86.9  2492.8   105.9 2495.42   139.2 2495.38   155.8 2492.46
   174.4 2492.58   276.1 2482.36   303.4  2480.9   315.9 2477.26   325.2 2476.16
   405.1 2475.26   422.7 2473.84   429.6 2472.19   436.6  2473.9   443.6 2475.99
   523.8 2474.01   571.2 2474.48   633.8 2476.94   643.7 2479.15   656.8 2483.94
   710.4  2510.5   723.2 2513.03   731.3 2516.22   829.8 2528.87   843.4 2529.76
     857 2528.84   872.9 2530.64   888.8 2533.93   902.4 2533.29     937  2534.4
#Mann= 8 ,-1 , 0
       0     .12       0      60      .1       0     110     .04       0
     240    .035       0   422.7    .045       0   436.6    .035       0
     630     .05       0     920      .1       0
#XS Ineff= 2 , 0
                          535.53         2478.59
Permanent Ineff=
       F       F
Bank Sta=422.7,436.6
XS Rating Curve= 0 ,0
Exp/Cntr(USF)=0,0
Exp/Cntr=0.3,0.1

Type RM Length L Ch R = 1 ,39514   ,174.7,186.3,186.5
XS GIS Cut Line= 4
2156304.47874691 241059.373359142156042.36541317241323.065688864
2155933.41469011241545.7041229432155715.51324399241743.078621239
#Sta/Elev= 30
       0 2517.92    77.4 2507.15   100.7 2500.16   119.3 2499.11     124 2496.49
   129.7 2491.95   147.3 2492.07     164 2490.14   175.2 2487.81   187.2 2483.62
   194.1 2482.55   310.1 2479.04     324 2477.68   414.4  2473.1   422.2    2472
   432.6 2470.86   440.42471.748   447.3 2473.14   474.4 2474.23   556.8 2474.02
   586.2 2475.64   643.7 2481.53     692 2484.37   740.9 2491.01     746 2492.74
   770.2 2497.43   809.3 2511.34     819 2516.01   877.7 2540.57   913.7 2553.94
#Mann= 7 ,-1 , 0
       0     .12       0      40     .04       0     270    .035       0
   422.2    .045       0   440.4    .035       0   511.8     .05       0
  819.67      .1       0
#XS Ineff= 2 , 0
                          456.58          2476.9
Permanent Ineff=
       F       F
Bank Sta=422.2,440.4
XS Rating Curve= 0 ,0
Exp/Cntr(USF)=0,0
Exp/Cntr=0.3,0.1

Type RM Length L Ch R = 1 ,39328   ,260.8,270.2,270.8
XS GIS Cut Line= 2
2156208.15999174240947.2646441072155595.50954903241597.810990493
#Sta/Elev= 30
       0 2516.43    39.6 2509.85    56.8  2508.6    87.5 2502.14   104.6 2497.54
   116.2 2490.78   133.4 2490.41   140.1 2489.04   163.1 2477.45   168.8 2476.37
   240.2 2474.68   356.2 2474.88     391 2471.59     429    2473   444.4 2470.06
   458.4 2469.04   465.1 2470.14   474.6 2472.45   565.1 2471.77     590 2473.71
   609.1 2482.01   625.5 2484.94   709.6 2510.33   741.5 2515.16   760.1 2522.58
   789.6 2529.92   803.1 2531.21   845.9 2542.45   884.2 2554.17   893.6 2555.41
#Mann= 6 ,-1 , 0
       0     .12       0      40     .04       0     180    .035       0
   444.4    .045       0   465.1    .035       0     610     .05       0
#XS Ineff= 2 , 0
                          482.89         2475.09
Permanent Ineff=
       F       F
Bank Sta=444.4,465.1
XS Rating Curve= 0 ,0
Exp/Cntr(USF)=0,0
Exp/Cntr=0.3,0.1

Type RM Length L Ch R = 1 ,39058   ,284,286.5,287.1
XS GIS Cut Line= 3
2156133.94718038240838.3139210482155595.50954903241198.325005941
 2155494.4538059241553.599102875
#Sta/Elev= 30
       0 2504.14    33.3 2503.34    61.8 2502.07    85.5 2500.86    96.9 2496.79
     109 2487.73   126.4 2487.42   144.4 2479.43   184.2 2475.22   203.9 2474.02
     271 2470.13   361.8 2470.95   428.9 2468.97   511.7 2470.64   534.7 2467.48
   543.3 2466.97   553.6 2467.82   574.9 2470.71   616.3  2470.2   658.9    2478
   718.2 2484.15   789.9 2501.08   810.3 2510.05   823.6 2512.37   868.3 2535.99
   878.6 2543.41   895.6 2545.93   908.6  2555.7     957 2578.51  1017.1 2599.97
#Mann= 9 ,-1 , 0
       0     .12       0    33.3      .1       0    61.8     .04       0
   184.2     .06       0   203.9    .035       0   534.7    .045       0
   553.6    .035       0   658.9     .05       0   908.6      .1       0
#XS Ineff= 2 , 0
          280.41    2480  601.24         2480.91
Permanent Ineff=
       F       F
Bank Sta=534.7,553.6
XS Rating Curve= 0 ,0
Exp/Cntr(USF)=0,0
Exp/Cntr=0.3,0.1

Type RM Length L Ch R = 1 ,38771   ,164.9,167.8,166.1
XS GIS Cut Line= 3
2156059.73436902240678.8353264242155361.81814305241008.845487576
2155178.65460863241379.909544374
#Sta/Elev= 30
       0 2510.88    36.4 2507.01      47 2508.86   123.4 2502.59   138.1 2492.12
     169 2491.98   203.4 2480.83   241.6 2479.73   256.4 2474.67   268.7 2472.86
   384.8 2467.92   395.7 2469.09   588.1 2468.98   591.5 2468.72   596.4 2465.21
   601.4 2464.38   609.8 2465.38   617.1 2468.65   630.9 2469.72   704.2 2469.27
   813.8 2471.61     889 2482.92   918.4 2491.25   942.9 2504.79   956.5 2508.89
  1007.7  2534.8  1097.2  2572.9  1154.1 2596.06  1172.4 2597.21  1185.8 2604.12
#Mann= 9 ,-1 , 0
       0      .1       0      80     .04       0     190      .1       0
     410    .035       0   596.4    .045       0   609.8    .035       0
  822.01      .1       0  922.01    .035       0  932.01      .1       0
Bank Sta=596.4,609.8
XS Rating Curve= 0 ,0
Exp/Cntr(USF)=0,0
Exp/Cntr=0.3,0.1

Type RM Length L Ch R = 1 ,38603   ,199.3,189,178.6
XS GIS Cut Line= 3
2155930.01115073240561.9305509612155321.73694188240855.580169028
2155123.63997731241326.351778945
#Sta/Elev= 30
       0 2507.37    49.2 2503.82    71.1 2498.83   114.8 2498.08   129.3  2490.3
   162.1  2486.2   180.3 2480.46   191.3 2480.28   224.1 2489.77   291.7 2485.28
   314.9 2478.83   341.9 2466.65   511.4 2467.76   519.2 2467.53   526.2 2464.56
   533.5 2463.01   544.92464.633     563 2467.69   588.4 2467.07   616.2    2469
   651.5 2468.02   825.5 2470.35   861.5  2473.3     889 2477.54   921.6 2487.22
   953.6 2501.36   967.8 2504.94     975 2509.71  1120.9 2571.43  1186.2 2592.61
#Mann= 10 ,-1 , 0
       0      .1       0      50     .04       0     160     .05       0
     270      .1       0     380    .035       0     490      .1       0
   526.2    .045       0   544.9      .1       0     600    .035       0
  995.45      .1       0
Bank Sta=526.2,544.9
XS Rating Curve= 0 ,0
Exp/Cntr(USF)=0,0
Exp/Cntr=0.3,0.1

Type RM Length L Ch R = 1 ,38414   ,437.9,436.5,436
XS GIS Cut Line= 2
     2155530.525      240322.147     2155125.822      241278.121
#Sta/Elev= 30
       0 2483.71    27.6 2477.14    48.9 2473.61   116.3 2472.66   130.9 2471.67
   141.6 2472.15   148.9 2470.83   159.4 2471.25     183 2469.77     219 2472.24
   234.2 2477.12   250.3    2477   258.7 2475.92   266.5 2473.67   280.5 2472.15
   317.6 2463.98   326.8 2462.97   337.5 2464.05   355.3 2464.76   371.6 2466.64
   460.7 2466.51   714.6 2469.88   772.2 2475.36   794.7 2479.46   817.2 2486.15
   832.7 2492.14   857.2 2503.34   868.4 2506.92  1007.4 2565.99  1038.1 2576.99
#Mann= 7 ,-1 , 0
       0      .1       0      40     .05       0      90      .1       0
   317.6    .045       0   337.5      .1       0     370    .035       0
     850      .1       0
Bank Sta=317.6,337.5
XS Rating Curve= 0 ,0
Exp/Cntr=0.3,0.1

Type RM Length L Ch R = 1 ,37978   ,376.9,379,376.5
XS GIS Cut Line= 2
     2155154.261      240204.017     2154795.497      241057.175
#Sta/Elev= 30
       0 2527.95   120.1 2517.87   191.3 2508.91   237.5 2499.06   251.8 2495.14
   262.5 2491.81   297.6 2477.57   319.4 2471.31   330.1 2469.83   345.3 2466.45
   365.7 2465.93   369.2 2464.95   376.4 2460.83   379.9 2459.96   390.6 2461.38
   427.92460.024   436.9 2458.89   440.4 2458.98   442.92460.152   447.5 2463.06
     449 2463.14   561.4 2463.62   583.3 2464.39   604.1  2466.1   636.2 2465.51
   652.2 2466.24   668.2 2467.99   703.8 2467.72   767.9 2468.66   925.5 2472.38
#Mann= 7 ,-1 , 0
       0    .035       0     170      .1       0     280    .035       0
   427.9    .045       0   442.9    .035       0     900     .05       0
     920      .1       0
#XS Ineff= 2 , 0
          380.76 2467.79  514.78         2468.96
Permanent Ineff=
       F       F
Bank Sta=427.9,442.9
XS Rating Curve= 0 ,0
Exp/Cntr=0.3,0.1

Type RM Length L Ch R = 1 ,37599   ,299.4,296.8,291
XS GIS Cut Line= 2
      2154802.06      240112.139     2154478.297      240952.171
#Sta/Elev= 30
       0  2522.9    48.3 2518.01    62.4 2515.25   143.3 2490.33   227.7 2474.58
   290.5  2467.1   326.1 2461.04   368.3 2460.31   378.82457.413   385.9 2455.54
   394.72457.398   402.1 2460.05   440.2  2460.8   554.7 2461.16   582.8  2459.6
   648.3 2461.85   663.7 2464.13   674.2 2462.33   681.1  2464.8   690.6 2471.75
   705.8 2480.33     727  2489.1     741 2500.19   790.2 2529.17   803.1 2532.91
   832.4 2551.58     843 2553.55   856.4 2562.36   867.6 2566.73   900.3 2582.87
#Mann= 8 ,-1 , 0
       0    .035       0      60      .1       0     370    .035       0
   378.8    .045       0   394.7    .035       0     690      .1       0
     810     .08       0     900      .1       0
#XS Ineff= 2 , 0
                          492.78         2476.36
Permanent Ineff=
       F       F
Bank Sta=378.8,394.7
XS Rating Curve= 0 ,0
Exp/Cntr=0.3,0.1

Type RM Length L Ch R = 1 ,37302   ,136.5,128.7,115.7
XS GIS Cut Line= 3
      2154666.43        240066.2     2154395.169       240282.77
     2154362.356      241022.174
#Sta/Elev= 30
       0 2521.16   107.6 2517.19     131 2515.64   156.9 2512.36     194  2505.1
   240.6 2494.16   347.1 2464.69   395.6 2463.22   424.22455.107   428.4 2454.17
   440.12455.223   448.1 2457.59   454.6  2458.1   526.9  2459.1     655 2458.06
   746.9 2459.95   756.8 2458.86   763.3 2460.22   779.8 2461.09   786.3 2463.48
   796.2 2465.21   812.6 2472.33   822.4 2479.08   948.7 2551.85   966.9 2563.26
   976.8  2565.4   989.9 2573.56  1026.1 2588.66  1042.5 2594.03  1087.2 2604.99
#Mann= 6 ,-1 , 0
       0    .035       0      80      .1       0     200    .035       0
   424.2    .045       0   440.1    .035       0  627.11      .1       0
#XS Ineff= 2 , 0
          391.58 2467.16  702.16         2461.41
Permanent Ineff=
       F       F
Bank Sta=424.2,440.1
XS Rating Curve= 0 ,0
Exp/Cntr=0.3,0.1

Type RM Length L Ch R = 1 ,37173   ,321.3,338.4,347.7
XS GIS Cut Line= 3
2153936.61189032240060.7899521512154353.17638856240498.053307453
2154335.06488864241010.350019582
#Sta/Elev= 30
       0  2475.9      22 2468.48    38.5 2464.91      80 2462.45    92.4 2463.27
   219.2 2457.76   314.5 2458.63   402.6 2456.07   480.8 2457.99   491.2 2454.18
   504.6 2455.47   513.8 2454.12   520.9 2452.91   527.9 2454.21     532 2457.21
   537.2 2457.89   599.9 2458.92   702.8 2457.67   774.9  2459.3   791.4 2458.03
   801.3 2459.99   824.3 2460.19   847.3 2464.29   857.1  2471.7   883.4 2486.14
    1018  2566.8  1031.1 2568.75  1047.8 2577.22  1067.2  2584.3  1116.5 2597.83
#Mann= 5 ,-1 , 0
       0      .1       0     140    .035       0   513.8    .045       0
   527.9    .035       0  663.92      .1       0
#XS Ineff= 2 , 0
          450.71 2460.38
Permanent Ineff=
       F       F
Bank Sta=513.8,527.9
XS Rating Curve= 0 ,0
Exp/Cntr(USF)=0,0
Exp/Cntr=0.3,0.1

Type RM Length L Ch R = 1 ,36835   ,303.7,302.9,301.9
XS GIS Cut Line= 3
2153918.54178642240089.1307139592154076.32917544240293.652094028
     2154049.531      241041.862
#Sta/Elev= 30
       0  2476.2    19.5 2468.05    44.6 2464.08   159.9 2460.26   196.5 2457.41
   258.1 2458.12   404.2 2456.31   476.4 2456.58   522.3 2454.87   538.8 2455.27
   551.9 2452.41   561.7 2454.19   581.4 2454.74     5952452.392   604.4 2450.37
   617.62452.146     634 2463.83   643.8 2464.94   647.1  2466.9   656.9 2475.86
   729.2 2518.41     739 2522.34   752.1 2530.18   771.8 2539.22   811.2 2553.57
   824.4 2559.57   834.2    2561   847.3 2566.71   899.9 2583.81    1007 2610.84
#Mann= 7 ,-1 , 0
       0      .1       0     100    .035       0     595    .045       0
   617.6    .035       0  628.31      .1       0  718.31     .08       0
  918.31      .1       0
#XS Ineff= 2 , 0
          511.11 2458.28
Permanent Ineff=
       F       F
Bank Sta=595,617.6
XS Rating Curve= 0 ,0
Exp/Cntr=0.3,0.1

Type RM Length L Ch R = 1 ,36532   ,346.1,350,351.6
XS GIS Cut Line= 3
     2153753.435      240179.426     2153762.719      240634.332
     2153772.004      241089.237
#Sta/Elev= 30
       0 2463.86    23.8 2460.65    76.3 2460.72   207.5 2456.03   266.6 2455.87
   315.8 2453.37   417.5 2453.76   429.9 2452.81   439.9 2450.83   453.6 2449.72
   463.6 2450.91     470 2453.69   483.2 2454.88   496.3 2461.31   506.1 2462.46
     516 2469.78   552.1 2487.04     575 2495.22   592.2 2500.15   604.6 2503.12
   627.6 2506.85   680.1 2512.81   709.6 2513.47   735.8 2512.69   762.7  2514.3
   791.6 2522.47     808 2529.37   867.1 2548.55   890.1 2556.89     910 2560.75
#Mann= 4 ,-1 , 0
       0    .035       0     380      .1       0   439.9    .045       0
   463.6      .1       0
#XS Ineff= 2 , 0
          350.11 2457.44
Permanent Ineff=
       F       F
Bank Sta=439.9,463.6
XS Rating Curve= 0 ,0
Exp/Cntr=0.3,0.1

Type RM Length L Ch R = 1 ,36182   ,351.8,350,347.7
XS GIS Cut Line= 3
     2153493.767      240149.689     2153419.787       240597.78
     2153367.589      241054.067
#Sta/Elev= 30
       0 2457.07    67.5  2456.6     132 2457.68   223.3 2456.62   257.1 2454.99
     267 2453.53   300.2 2451.34   366.8  2450.9     430  2452.4   433.3 2452.11
   441.8  2448.8   449.9 2446.88   469.8 2448.74   479.7 2449.54   486.3 2451.95
   499.5 2454.31   509.4 2458.67   525.6 2469.28   548.6  2479.8   572.1 2488.73
   595.2 2495.81   614.5 2502.82     668 2515.23   700.4 2524.67   746.3 2536.66
   763.7 2542.14   780.4 2545.88   796.7 2548.26   842.9 2559.21   913.4  2572.5
#Mann= 5 ,-1 , 0
       0      .1       0      20    .035       0   441.8    .045       0
   469.8    .035       0  514.16      .1       0
Bank Sta=441.8,469.8
XS Rating Curve= 0 ,0
Exp/Cntr=0.3,0.1
